HEC-RAS study TRKYCK.prj: TRKYCK

--- TRKYCK.g01 (geometry) --- (continued)

Type RM Length L Ch R = 1 ,18172.6 ,186.7,183.6,180.1
XS GIS Cut Line= 3
     2102733.296      194545.663     2102528.802      194907.459
     2102643.386      195074.805
#Sta/Elev= 30
       0 1927.49    13.1 1925.11    42.5 1921.13    65.4 1919.24    88.4 1918.27
   134.2 1912.75   206.2 1907.23  218.231905.127  237.271902.614  282.321901.285
   294.5  1899.4   310.9 1898.92   317.4 1897.88     324 1896.23   330.5 1896.11
     337  1896.3   343.6 1897.86   350.1 1898.97   353.4  1900.1   366.5 1905.51
   379.6 1911.75   405.8 1921.82   415.6  1923.4   435.2 1928.56   451.6 1932.19
   464.7 1934.41   484.3 1939.39   549.7 1952.81   585.7 1959.56   618.4 1964.12
#Mann= 6 ,-1 , 0
       0     .06       0  218.23     .12       0  237.27     .06       0
  282.32    .016       0   317.4    .045       0   343.6     .12       0
#XS Ineff= 2 , 0
          282.46 1903.51
Permanent Ineff=
       F       F
Bank Sta=317.4,343.6
XS Rating Curve= 0 ,0
Exp/Cntr=0.3,0.1

Type RM Length L Ch R = 1 ,17989   ,36,37.4,40.2
XS GIS Cut Line= 4
     2102127.669      194560.253     2102409.227      194744.048
     2102364.957      194859.933     2102597.818      195115.582
#Sta/Elev= 30
       0 1995.35    29.4 1988.09      62 1977.88    94.7 1970.51   104.5 1967.29
  143.241957.315  177.411947.913   199.1 1940.06  209.521937.479   231.8 1929.68
     271 1913.58  296.781901.745   303.6  1900.2   323.2  1901.2   336.2 1899.63
     346 1899.54  361.411895.295   368.9 1894.48   383.51895.081  403.79 1896.87
   440.7 1899.09   460.3 1901.38   476.6 1906.37     506 1911.98   584.3 1924.34
   659.3 1938.52   711.5 1945.83   737.6  1950.5     767 1952.87   806.1 1952.96
#Mann= 8 ,-1 , 0
       0     .06       0  143.24     .12       0  177.41     .06       0
  209.52     .12       0  296.78    .016       0  361.41    .045       0
   383.5    .016       0  403.79     .12       0
#XS Ineff= 2 , 0
                          405.57         1902.09
Permanent Ineff=
       F       F
Bank Sta=361.41,383.5
XS Rating Curve= 0 ,0
Exp/Cntr=0.3,0.1

Type RM Length L Ch R = 1 ,17951.6 ,369.1,328.9,286.8
XS GIS Cut Line= 4
     2102118.576      194569.933     2102374.505      194739.707
     2102330.234      194855.593     2102585.156      195130.914
#Sta/Elev= 30
       0 1995.11    26.1 1988.74    65.3 1976.29  145.481956.688   173.2 1949.48
   189.5 1943.89   215.6 1937.38   284.2 1906.26  299.821901.482   307.1  1899.4
   323.4  1898.5   339.9 1894.55   349.6 1893.74   365.9 1894.44   369.2 1894.13
   385.5 1897.65   408.3 1898.78   421.4 1897.81   431.2 1898.11   437.7 1900.12
     454 1900.23  462.391901.868   473.6 1905.39   496.4  1909.5   561.7 1919.56
   574.7 1922.66   613.9 1929.43     715 1945.57   760.7 1948.29   806.4 1947.64
#Mann= 6 ,-1 , 0
       0     .06       0  145.48     .12       0  299.82    .016       0
   339.9    .045       0   365.9    .016       0  462.39     .12       0
#XS Ineff= 2 , 0
          319.92 1901.49  402.48         1901.89
Permanent Ineff=
       F       F
Bank Sta=339.9,365.9
XS Rating Curve= 0 ,0
Exp/Cntr=0.3,0.1

Type RM Length L Ch R = 1 ,17622.6 ,146.9,143.7,140.5
XS GIS Cut Line= 3
     2102009.368      194996.994     2102319.167      195066.313
     2102502.742       195201.76
#Sta/Elev= 30
       0 1989.33    22.9 1976.07    65.5 1957.04   104.7 1938.42   117.8 1930.41
   134.2 1921.84   153.8 1908.01   176.7 1895.34   196.4 1888.48     2021887.724
   223.21887.595   232.4 1887.41   238.9 1888.49   245.5  1891.9     252 1894.04
   281.5 1897.19  296.241897.916   301.1 1898.76   307.6 1901.78   310.9  1902.3
   327.2  1902.4   343.5 1906.04   353.3  1906.2  360.651907.127   379.4 1910.55
   428.3  1914.5   486.9 1917.92   519.5 1920.94   532.6 1922.68   545.6 1927.34
#Mann= 5 ,-1 , 0
       0     .12       0     202    .045       0   223.2     .12       0
  296.24    .016       0  360.65     .12       0
Bank Sta=202,223.2
XS Rating Curve= 0 ,0
Exp/Cntr=0.3,0.1

Type RM Length L Ch R = 1 ,17478.9 ,251.9,250.8,249.8
XS GIS Cut Line= 3
     2101989.007      195168.838      2102302.24      195191.313
     2102480.966      195314.866
#Sta/Elev= 30
       0 1998.89    32.7 1984.93    45.8 1976.72    62.2 1968.47      85 1953.44
    98.1  1942.9   104.7 1938.69   176.6 1894.76     193 1886.62   199.5 1886.08
   215.9 1886.37     229 1888.16   251.9 1888.64   261.7 1892.12   281.3 1893.34
   291.1 1895.59  324.361900.012     340 1906.43  344.721907.051   365.9 1906.56
   377.51911.246   391.9 1916.37   424.3 1923.77   430.8 1924.27     4501929.371
   476.2 1931.96  486.341937.537   492.4 1940.45   515.1  1946.4   531.3 1952.23
#Mann= 8 ,-1 , 0
       0     .12       0     193    .045       0   215.9     .12       0
  324.36     .08       0  344.72    .016       0   377.5     .12       0
     450    .016       0  486.34     .12       0
Bank Sta=193,215.9
XS Rating Curve= 0 ,0
Exp/Cntr=0.3,0.1

Type RM Length L Ch R = 1 ,17228.1 ,168.9,141.4,116
XS GIS Cut Line= 3
     2101958.269      195428.268     2102196.634      195432.171
     2102470.847      195441.352
#Sta/Elev= 30
       0 2000.46    45.7 1982.44      62 1973.22    71.8 1969.82    94.7 1954.93
   133.9 1933.93   153.5 1918.96   179.6 1902.19   195.9 1894.01     209 1891.25
   218.8 1885.67   225.3 1884.18   238.4  1883.9   244.9 1884.13   264.5 1889.77
  311.091893.007   326.6 1898.84     356 1901.04  365.811906.704   382.1  1912.6
   408.2    1926   434.4 1933.77   444.2  1937.4  455.751943.241   463.8 1946.78
   480.1 1947.36   483.4 1948.41  486.531951.061   493.2  1956.1   512.8 1963.98
#Mann= 7 ,-1 , 0
       0     .12       0   225.3    .045       0   244.9     .12       0
  311.09    .016       0  365.81     .12       0  455.75    .016       0
  486.53     .12       0
Bank Sta=225.3,244.9
XS Rating Curve= 0 ,0
Exp/Cntr=0.3,0.1

Type RM Length L Ch R = 1 ,17086.7 ,59.5,57.9,58
XS GIS Cut Line= 4
     2101927.604      195524.794     2102166.319      195607.259
     2102234.679       195530.22     2102469.054      195516.114
#Sta/Elev= 30
       0 2006.17    91.8 1962.77   160.7 1923.71     187 1911.31   209.9 1897.54
   219.8  1894.2   229.6 1892.78  249.971893.337   255.8 1893.65   265.4 1887.98
   284.7 1883.22   300.8 1882.81   310.5 1883.23   323.4 1883.96   329.8 1886.52
   336.2 1893.51   342.7 1895.28  400.821896.563     411 1897.77  418.391900.696
   427.3 1905.23   448.5 1907.36   482.7 1924.32   531.6 1944.13  538.231948.661
   551.2  1955.1   564.3 1955.32  568.931956.701   580.6 1964.49   590.4 1969.36
#Mann= 9 ,-1 , 0
       0     .12       0  249.97    .016       0   284.7    .045       0
   310.5    .016       0  400.82     .12       0  418.39    .016       0
   448.5     .12       0  538.23    .016       0  568.93     .12       0
Bank Sta=284.7,310.5
XS Rating Curve= 0 ,0
Exp/Cntr=0.3,0.1

Type RM Length L Ch R = 1 ,17028.8 ,257.7,299.4,338.3
XS GIS Cut Line= 4
     2101908.073      195569.282     2102169.575      195660.428
     2102237.934      195583.388     2102472.309      195569.282
#Sta/Elev= 30
       0  2005.6    78.2 1971.92   153.1 1932.72   175.9  1917.9   228.1 1894.52
  237.271892.476   267.2 1892.98   270.4 1892.11   276.9 1885.92   280.2 1884.65
   302.7 1882.38   309.1 1881.69   328.4 1882.18   344.5 1883.28  353.091885.748
   379.9 1890.64   412.5 1892.26   428.8 1897.06  437.371901.542   451.7 1903.58
  471.731910.177   484.3 1914.64   507.1 1927.93   536.5 1938.77  561.461951.403
   575.6  1959.8  592.151960.854   595.2 1961.51   604.9  1969.5   614.7 1974.93
#Mann= 9 ,-1 , 0
       0     .12       0  237.27    .016       0   302.7    .045       0
   328.4    .016       0  353.09     .12       0  437.37    .016       0
  471.73     .12       0  561.46    .016       0  592.15     .12       0
Bank Sta=302.7,328.4
XS Rating Curve= 0 ,0
Exp/Cntr=0.3,0.1

Type RM Length L Ch R = 1 ,16729.4 ,269.9,278.7,284.2
XS GIS Cut Line= 3
     2101814.377      195743.405     2102130.716      195915.774
     2102324.871      196061.385
#Sta/Elev= 30
       0 1963.05    45.8 1957.52   74.261951.858   104.8 1942.76   147.4 1925.73
   173.6 1912.96     190 1902.13  192.371899.486   196.5 1895.18     203 1891.47
   222.7 1891.21     226 1890.41  235.711884.582   245.6  1882.1     262 1883.49
   278.4  1881.5   314.4 1882.34   337.3 1881.65   353.7 1879.61   363.5 1879.06
   373.4 1879.64   389.8 1880.97   399.6 1883.01   412.7 1888.49   425.8 1897.33
   461.9  1924.3   494.7 1944.62   550.5 1976.68  595.862000.224   602.9 2004.57
#Mann= 7 ,-1 , 0
       0     .06       0   74.26     .12       0  192.37    .016       0
  235.71     .12       0   353.7    .045       0   373.4     .12       0
  595.86    .016       0
#XS Ineff= 2 , 0
          265.12 1887.57
Permanent Ineff=
       F       F
Bank Sta=353.7,373.4
XS Rating Curve= 0 ,0
Exp/Cntr=0.3,0.1

Type RM Length L Ch R = 1 ,16450.7 ,213.2,223.1,228.5
XS GIS Cut Line= 3
     2101734.518       195867.13     2101919.095      196092.039
     2102053.185      196258.358
#Sta/Elev= 30
       0 1935.13    13.1 1932.58    65.4 1924.81   101.3 1917.59   124.2 1910.73
   143.8 1908.04   153.6 1904.11     1671895.835   173.3 1891.77   176.5 1890.95
   199.4 1891.35   202.7 1890.22  205.951888.162   212.5 1883.82   215.8 1882.58
   251.7  1881.5   274.6 1878.58   294.2 1877.39   307.1 1877.31   316.8 1877.31
   329.8 1878.87   349.2 1878.14   365.4 1882.97   384.8 1893.44   394.5 1896.14
     401  1900.2   410.7 1905.04   420.4    1911   446.3 1925.34   504.6  1955.9
#Mann= 5 ,-1 , 0
       0     .12       0     167    .016       0  205.95     .12       0
   294.2    .045       0   316.8     .12       0
#XS Ineff= 2 , 0
          252.63 1883.65
Permanent Ineff=
       F       F
Bank Sta=294.2,316.8
XS Rating Curve= 0 ,0
Exp/Cntr=0.3,0.1

Type RM Length L Ch R = 1 ,16227.6 ,239.7,250,267.5
XS GIS Cut Line= 3
     2101652.747       195906.74     2101728.713      196202.542
     2101813.497      196386.854
#Sta/Elev= 30
       0 1927.34      13 1925.51    29.2 1921.16    45.5 1920.07      65 1915.41
      91 1913.34   136.5 1907.62     143 1905.28  150.291901.139   162.4 1899.18
   188.4 1898.79  194.151897.607   214.4 1889.35   227.4 1886.64   240.4 1882.15
   266.4 1879.81   279.4  1875.8   294.61873.223   311.9 1873.12   316.21873.184
   328.3 1874.65   331.6 1876.08   344.7 1889.39   354.5  1895.7   377.4 1908.57
   400.3 1920.15     433 1938.93   446.1 1944.82   472.3 1962.79   508.3 1980.49
#Mann= 5 ,-1 , 0
       0     .12       0  150.29    .016       0  194.15     .12       0
   294.6    .045       0   316.2     .12       0
Bank Sta=294.6,316.2
XS Rating Curve= 0 ,0
Exp/Cntr=0.3,0.1

Type RM Length L Ch R = 1 ,15977.6 ,239.3,249.4,251.6
XS GIS Cut Line= 3
     2101551.115      195911.952     2101486.437      196230.363
     2101426.715      196396.257
#Sta/Elev= 30
       0 1922.13   42.371914.384   66.081909.351    71.5 1908.44    81.2 1904.47
    84.5 1903.69     104 1903.07  116.971899.188   126.7 1896.34   152.7 1890.35
  175.481885.786   214.4 1880.32   295.7 1873.36  302.811871.863   311.9 1870.47
   324.9 1870.22   331.4 1870.37   334.7 1870.87     338 1872.65   354.3 1886.11
   364.1 1894.92   373.9 1900.48     387 1910.39   403.3 1920.26   419.6 1931.65
   429.4 1939.04   458.8 1958.56   465.3 1962.08   478.4 1967.73   501.2 1976.15
#Mann= 8 ,-1 , 0
       0     .06       0   42.37     .12       0   66.08    .016       0
  116.97     .12       0  175.48     .06       0  302.81     .12       0
   311.9    .045       0   331.4     .12       0
Bank Sta=311.9,331.4
XS Rating Curve= 0 ,0
Exp/Cntr=0.3,0.1

Type RM Length L Ch R = 1 ,15728.2 ,263.3,250.3,240.2
XS GIS Cut Line= 3
     2101428.812      195904.551     2101278.005      196099.131
     2101176.034      196307.693
#Sta/Elev= 30
       0 1914.04    6.991913.376   16.531912.095    25.9 1911.07    35.6 1906.41
    55.1 1905.34    58.3  1904.3    64.8 1900.73   71.361898.667    84.2 1895.87
     162 1876.25   204.1 1870.68     217  1870.5     230 1868.31   239.7 1868.02
   242.9    1868   262.5 1868.16   265.8 1869.27   269.1 1871.83   275.6 1879.45
   285.4 1887.32   311.6 1900.97   334.5 1908.23   344.3 1912.38   354.1 1915.42
   399.9 1926.79   422.8 1930.97   442.4  1933.6   458.7 1938.13   478.3 1944.53
#Mann= 6 ,-1 , 0
       0     .06       0    6.99     .12       0   16.53    .016       0
   71.36     .12       0   239.7    .045       0   262.5     .12       0
Bank Sta=239.7,262.5
XS Rating Curve= 0 ,0
Exp/Cntr=0.3,0.1

Type RM Length L Ch R = 1 ,15477.9 ,256,250,248.3
XS GIS Cut Line= 3
     2101063.351      195774.639     2101052.051      196006.309
     2101046.646      196277.462
#Sta/Elev= 30
       0 1925.08    9.241921.439    13.1 1920.23    42.5 1919.22   47.071917.998
    75.1 1909.69   104.5 1902.72   127.4 1896.07  135.341894.776   140.5 1893.84
   143.7 1892.29   150.3 1887.11   153.5 1885.57   176.4 1882.98  185.421878.711
   199.3 1871.15  220.131866.325   228.7 1865.55   241.8 1866.26   258.1 1869.26
   271.2 1868.39   284.2 1871.01   310.4 1872.74   316.9  1873.8   333.2 1878.51
   349.6 1885.06   372.4 1898.05   441.1 1928.72   463.9 1939.69   503.2 1955.84
#Mann= 7 ,-1 , 0
       0     .12       0    9.24    .016       0   47.07     .12       0
  135.34    .016       0  185.42     .12       0  220.13    .045       0
   241.8     .12       0
Bank Sta=220.13,241.8
XS Rating Curve= 0 ,0
Exp/Cntr=0.3,0.1

Type RM Length L Ch R = 1 ,15227.9 ,247.3,250,246.9
XS GIS Cut Line= 3
     2100757.681      195788.807     2100830.211      196101.256
     2100835.789      196271.659
#Sta/Elev= 30
       0 1931.24    26.2 1923.32    94.9 1904.71  149.621891.864   189.8 1878.56
   196.4 1877.11   208.11876.334  245.541874.235   255.3 1872.68   258.6 1871.79
   265.1 1868.96   281.5 1868.34  287.351867.376   309.91864.667   314.2 1864.03
     324 1863.75   330.6 1863.96   333.9 1864.55   340.4 1866.62   350.3 1871.44
   360.1 1877.79   369.9 1885.14     383 1893.59   392.9 1899.13   399.4 1903.93
   419.1 1913.52   438.8 1924.56   458.5 1934.86   471.6 1940.37   491.2 1949.76
#Mann= 7 ,-1 , 0
       0     .12       0  149.62     .06       0   208.1     .12       0
  245.54    .016       0  287.35     .12       0   309.9    .045       0
   333.9     .12       0
Bank Sta=309.9,333.9
XS Rating Curve= 0 ,0
Exp/Cntr=0.3,0.1

Type RM Length L Ch R = 1 ,14977.9 ,236.4,241.5,247.1
XS GIS Cut Line= 3
     2100543.791      195810.376     2100581.568      196103.792
     2100612.386      196292.164
#Sta/Elev= 30
       0 1919.52    29.3 1913.41      78 1901.48   99.551896.535   126.8 1890.77
  163.881885.074   172.3 1883.72   185.3 1881.03   204.8 1878.02   247.1 1868.53
  256.981864.617   263.3 1863.87   276.3 1864.02  287.911862.326   292.6 1861.75
   295.8 1861.73     312 1862.27   318.5 1862.76     325 1863.83   337.9 1868.18
   344.4 1871.11   370.2 1883.43   386.4 1892.36   396.1 1898.69   409.1 1904.85
   428.5 1915.77   441.4 1922.51   460.8  1931.7     477 1938.71   486.7 1942.49
#Mann= 6 ,-1 , 0
       0     .06       0   99.55     .12       0  163.88     .06       0
  256.98    .016       0  287.91    .045       0     312     .12       0
Bank Sta=287.91,312
XS Rating Curve= 0 ,0
Exp/Cntr=0.3,0.1

Type RM Length L Ch R = 1 ,14736.4 ,211.3,206,200
XS GIS Cut Line= 3
     2100376.871      195827.208        2100340.      196190.011
     2100418.075      196335.182
#Sta/Elev= 30
       0 1914.26    48.8 1901.98   107.4 1889.39  142.211878.337  152.881875.017
   166.1 1870.92  179.18 1868.58   185.6 1867.26   198.6 1866.24  254.881863.287
   263.7 1863.01   273.5 1861.43  285.62 1862.33     293 1861.95   299.6 1861.23
   312.6 1861.42   315.8 1861.98   319.1 1862.91   341.9 1862.98   348.4  1864.4
   358.2  1869.7   367.9 1873.53   390.5 1885.56   419.6  1899.4   445.5 1910.02
   471.3 1922.46   477.8 1926.09   503.6 1937.13   519.8  1942.9   529.5 1944.99
#Mann= 8 ,-1 , 0
       0     .06       0  142.21     .12       0  152.88     .06       0
  179.18     .12       0  254.88    .016       0  285.62     .12       0
     293    .045       0   315.8     .12       0
Bank Sta=293,315.8
XS Rating Curve= 0 ,0
Exp/Cntr=0.3,0.1

Type RM Length L Ch R = 1 ,14530.4 ,321.3,303.6,280.3
XS GIS Cut Line= 3
     2100113.372      195903.674     2100174.635      196296.782
      2100311.65      196392.804
#Sta/Elev= 30
       0 1921.85    26.1 1912.46    42.4 1905.67    58.7 1898.73    78.3 1887.72
   120.7 1870.52   140.2  1864.8  170.751861.535   198.9 1861.27  203.781860.519
  207.171859.892     225 1859.33  230.011859.834   247.8 1861.91   273.9  1860.9
     287 1862.05   303.3 1867.89   313.1 1872.82   326.1 1880.96   358.7 1894.63
   397.8 1902.44   407.7 1905.64   433.9 1911.96   466.8 1916.82     493 1923.93
   519.2 1929.84   532.4 1932.29   545.5  1933.1   558.6 1936.26   565.2 1937.01
#Mann= 5 ,-1 , 0
       0     .12       0  170.75    .016       0  203.78     .12       0
  207.17    .045       0  230.01     .12       0
Bank Sta=207.17,230.01
XS Rating Curve= 0 ,0
Exp/Cntr=0.3,0.1

Type RM Length L Ch R = 1 ,14226.8 ,263.8,249.5,242.3
XS GIS Cut Line= 3
     2099751.034      196134.575     2099901.441      196258.011
     2100265.769      196429.508
#Sta/Elev= 30
       0 1990.22    16.2 1980.55    32.4 1974.58    42.2 1969.34    45.4 1966.53
    51.9 1958.01    58.4 1951.98    81.1 1934.68      94  1927.2     107 1916.04
   129.7 1900.14   158.9 1882.38   165.4 1876.92   171.9 1868.64   181.6  1859.5
   188.1 1857.38   201.1 1856.64   214.2 1857.58   220.8 1859.26   250.2 1858.12
   273.1 1859.51   305.9    1875  316.041877.066   341.9 1885.65   413.9 1900.28
   440.1 1903.12   456.5 1907.76  469.871909.839  512.261918.543   597.2 1931.71
#Mann= 6 ,-1 , 0
       0     .12       0   188.1    .045       0   214.2     .12       0
  316.04     .06       0  469.87     .12       0  512.26     .06       0
Bank Sta=188.1,214.2
XS Rating Curve= 0 ,0
Exp/Cntr=0.3,0.1

Type RM Length L Ch R = 1 ,13977.3 ,256.9,246.7,231.1
XS GIS Cut Line= 3
     2099617.674      196495.922     2099814.689      196489.473
      2100252.86       196555.52
#Sta/Elev= 30
       0 1949.79    16.2 1941.22      42 1930.15    64.6 1917.06    80.8 1908.99
   135.7    1884   155.1    1871   177.7 1858.71   190.7 1854.54   197.1 1854.27
   210.2 1854.51   219.9 1856.35   275.3 1858.82   278.6 1859.88   288.4 1865.49
   298.1 1868.95   337.2 1880.41   363.3 1886.55   376.3 1887.91  393.621891.516
  395.331891.826  431.941898.178   467.6 1904.03   483.8 1905.76  497.461908.658
   545.8 1917.83     562 1921.86   581.6 1927.52   610.9 1938.34   640.2 1946.64
#Mann= 7 ,-1 , 0
       0     .12       0   190.7    .045       0   210.2     .12       0
  393.62     .06       0  395.33     .12       0  431.94     .06       0
  497.46     .12       0
Bank Sta=190.7,210.2
XS Rating Curve= 0 ,0
Exp/Cntr=0.3,0.1

Type RM Length L Ch R = 1 ,13730.6 ,341.3,328,313.5
XS GIS Cut Line= 3
     2099685.433       196819.94     2099991.042      196653.553
     2100280.027      196628.529
#Sta/Elev= 30
       0 1974.23      13 1962.11    35.8 1946.55    55.3 1934.82    71.5 1922.64
   107.3 1899.94   123.6 1888.38   143.1 1873.01   156.1 1864.08   165.8 1858.73
   175.6 1854.54   182.1 1852.66   191.41851.789   198.4 1851.49   211.4 1851.79
   221.1 1854.42   234.2  1854.9   247.2  1857.3   273.2 1858.54   286.2 1858.29
   331.7 1871.98   351.2 1876.19   396.8 1887.73     449 1903.97   475.1 1910.32
   484.8 1913.69   533.7 1927.42   572.8 1937.17   615.2 1945.68     638 1952.69
#Mann= 3 ,-1 , 0
       0     .12       0   191.4    .045       0   211.4     .12       0
Bank Sta=191.4,211.4
XS Rating Curve= 0 ,0
Exp/Cntr=0.3,0.1

Type RM Length L Ch R = 1 ,13402.5 ,163.2,175.4,185.7
XS GIS Cut Line= 4
     2099917.665       197018.26     2100113.437      196894.438
     2100178.542       196764.23     2100349.572      196710.543
#Sta/Elev= 30
       0 1936.69      13 1932.19    42.4 1924.22    81.6 1907.67   127.2 1894.87
     137 1890.84   146.8 1885.86   156.6 1882.61   166.4 1877.69  189.531869.121
  205.621863.083   225.1 1857.06   247.8 1852.13   260.8 1851.13   273.7 1851.39
   287.11849.449   299.6 1848.78   309.21849.638   312.5 1850.97   322.2 1857.02
   328.7 1859.17   354.6 1872.99   364.3 1879.87     387 1892.68   396.8  1896.5
   439.2 1916.35   465.2 1931.17   514.1 1952.72     550 1966.98   556.5 1968.96
#Mann= 5 ,-1 , 0
       0     .12       0  189.53     .06       0  205.62     .12       0
   287.1    .045       0   309.2     .12       0
Bank Sta=287.1,309.2
XS Rating Curve= 0 ,0
Exp/Cntr=0.3,0.1

Type RM Length L Ch R = 1 ,13227.1 ,242.3,251.9,270.7
XS GIS Cut Line= 3
     2100013.353      197105.504     2100266.563      196953.754
     2100436.578      196826.241
#Sta/Elev= 30
       0 1923.53    29.5 1913.28    72.2  1902.2    95.1 1894.41   121.4 1886.62
   137.8    1880   154.2 1876.04   190.2 1864.03   226.3  1854.2   232.9 1853.16
   259.1 1852.22   272.2  1850.2   282.1 1849.54   291.9 1847.22   298.5 1846.94
   314.8 1847.24   318.1 1848.15   321.4 1850.62   327.9 1860.22   331.2 1863.16
   347.5  1874.6   373.7 1891.02   396.6 1906.56   406.4 1912.26   416.2 1919.65
   432.5 1930.76   445.6 1944.69   458.7    1951   484.8  1965.8   507.7 1976.04
#Mann= 3 ,-1 , 0
       0     .12       0   291.9    .045       0   314.8     .12       0
Bank Sta=291.9,314.8
XS Rating Curve= 0 ,0
Exp/Cntr=0.3,0.1

Type RM Length L Ch R = 1 ,12975.2 ,189.5,196.7,195.4
XS GIS Cut Line= 3
     2100060.425      197221.756     2100261.488      197186.656
      2100521.29      197237.668
#Sta/Elev= 30
       0 1913.29    29.2 1904.84    48.6 1897.21    77.8    1888   103.7  1882.9
   129.6 1876.32   158.8 1864.53   168.5 1857.15   178.2 1855.33   181.4 1853.61
   184.7 1849.74   187.9 1847.07   191.1 1845.63   200.9 1845.09  212.391845.565
   220.4 1847.24   230.2 1847.22   253.1 1848.92   279.3 1848.56   289.1 1850.16
   298.9 1855.56   305.4  1861.8   321.8 1872.65   331.6  1881.3   344.7  1888.9
   354.5 1896.26   387.2 1914.23   416.6 1929.44   449.2 1949.18   468.9 1957.91
#Mann= 3 ,-1 , 0
       0     .12       0   191.1    .045       0  212.39     .12       0
Bank Sta=191.1,212.39
XS Rating Curve= 0 ,0
Exp/Cntr=0.3,0.1

Type RM Length L Ch R = 1 ,12778.5 ,289.2,303.6,320.2
XS GIS Cut Line= 2
     2100078.678      197355.406     2100488.566       197416.01
#Sta/Elev= 30
       0 1902.89    19.6 1895.96    71.8 1881.25    81.6 1877.02   110.9 1868.44
   127.2 1861.12   133.8 1859.09   146.8 1852.63   159.9 1851.35   169.6 1846.22
  178.681843.304   189.2 1842.96   202.3 1843.23   208.8 1845.73   218.6 1846.34
   238.2 1849.63   257.7 1851.32   264.3 1852.89   267.5 1854.68     274 1860.44
   283.8 1866.83   303.4 1881.28   319.7 1888.56   326.3 1890.77     336 1897.29
   368.7 1910.03   381.7 1916.18   394.8 1920.59   404.6 1927.07   414.3 1932.07
#Mann= 3 ,-1 , 0
       0     .12       0  178.68    .045       0   202.3     .12       0
Bank Sta=178.68,202.3
XS Rating Curve= 0 ,0
Exp/Cntr=0.3,0.1

Type RM Length L Ch R = 1 ,12475   ,248.1,251.7,251.8
XS GIS Cut Line= 3
     2099978.237      197501.833     2100131.424      197632.909
     2100289.572      197829.725
#Sta/Elev= 30
       0 1905.67      26 1896.78      52 1884.88    61.8 1880.94      78 1873.17
    97.6 1866.72   110.6 1861.84   133.3 1852.27   149.6 1846.48   152.8 1845.77
   162.6 1845.64   175.6 1843.79   188.6 1843.23   198.4 1840.88   201.6 1840.61
   208.2 1840.47     218 1840.57   227.8 1842.58     241  1844.2   247.5 1846.21
   257.4 1851.44   270.5 1859.88     277 1864.95   283.6 1867.95   306.5 1880.09
   326.2 1888.31   345.9 1898.07   375.4 1909.57   424.6 1930.42   454.1 1939.52
#Mann= 3 ,-1 , 0
       0     .12       0   201.6    .045       0     218     .12       0
Bank Sta=201.6,218
XS Rating Curve= 0 ,0
Exp/Cntr=0.3,0.1

Type RM Length L Ch R = 1 ,12223.3 ,240.5,251.7,259.9
XS GIS Cut Line= 3
     2099817.735       197627.66     2099929.193      197776.744
     2100081.814      197973.546
#Sta/Elev= 30
       0 1912.47    19.6 1906.11    35.9 1899.75    45.7  1894.3    55.5 1888.03
    75.1 1878.05    84.9 1871.84   114.3 1855.44   120.8  1852.4   127.4 1850.01
   133.9 1846.52   137.2 1845.45   166.6 1841.34  184.961837.781   192.7 1837.53
  200.751837.738   205.8  1838.5   212.4 1840.56   222.2 1841.84     232 1842.33
     255 1842.14   261.5    1844   268.1 1846.55   277.9  1851.3   287.7 1856.99
   294.3 1862.27   300.8 1866.04     327 1877.75     386 1899.61   435.2 1915.46
#Mann= 3 ,-1 , 0
       0     .12       0  184.96    .045       0  200.75     .12       0
Bank Sta=184.96,200.75
XS Rating Curve= 0 ,0
Exp/Cntr=0.3,0.1

Type RM Length L Ch R = 1 ,11971.6 ,239.2,250,262.6
XS GIS Cut Line= 3
     2099666.813      197649.864     2099706.842      197886.067
     2099771.341      198111.818
#Sta/Elev= 30
       0 1920.84    19.4 1913.51    42.1 1907.04    77.7 1894.79   119.8 1879.67
   139.2 1871.59   155.4    1866   168.4 1859.78   171.6 1857.56   178.1 1850.78
   181.3 1848.32     191 1846.14   194.2 1844.61   200.7 1840.26     204 1839.18
   220.2 1838.31   229.9 1836.14   233.1 1836.08   252.6 1836.24   259.1 1838.32
   262.4 1838.79   278.7  1839.1     295 1839.89   298.3 1840.51   314.6 1848.96
   337.4 1862.59   376.5  1887.6   435.2 1920.07   461.3 1935.86   474.4 1942.39
#Mann= 3 ,-1 , 0
       0     .12       0   229.9    .045       0   252.6     .12       0
Bank Sta=229.9,252.6
XS Rating Curve= 0 ,0
Exp/Cntr=0.3,0.1

Type RM Length L Ch R = 1 ,11721.6 ,246.5,250,253.7
XS GIS Cut Line= 3
     2099527.473      197645.425     2099463.447      197856.713
     2099404.434      198051.459
#Sta/Elev= 30
       0 1918.18    35.7 1905.98    71.4  1891.9   110.4 1873.25   123.4 1868.36
   142.9 1859.55   149.4  1855.9   155.8  1851.3   172.1 1840.94   175.3 1839.74
   185.1 1838.28   191.6 1836.38   201.3 1835.26  206.771833.715   217.5 1833.13
   227.2  1833.5   243.4 1836.96   275.7 1835.97   278.9 1836.19   285.4 1838.29
   295.1 1843.23   320.9 1859.24   333.8 1865.87   359.7 1881.56   372.6 1890.83
   375.8 1893.68   382.3 1901.66   385.5 1904.33     421 1924.96   424.3 1926.49
#Mann= 3 ,-1 , 0
       0     .12       0  206.77    .045       0   227.2     .12       0
Bank Sta=206.77,227.2
XS Rating Curve= 0 ,0
Exp/Cntr=0.3,0.1

Type RM Length L Ch R = 1 ,11471.6 ,253.3,250,246
XS GIS Cut Line= 3
     2099322.691      197585.697     2099225.215      197788.811
     2099147.466       197944.31
#Sta/Elev= 30
       0 1932.79     9.8 1926.94    19.6 1921.72    32.6 1915.52    52.2 1906.77
    71.8 1898.72    84.9 1892.54      98 1887.68   114.3 1878.96   133.9 1867.41
   146.9    1858     160 1847.41   166.5 1843.05     173  1838.1   176.3 1836.53
   179.6 1835.63   192.6 1834.18     209 1833.43   215.5 1831.88     222 1831.46
   239.5 1831.84   254.8 1834.47   258.1 1835.32   264.7 1838.28   297.5 1856.54
     304 1860.64   340.1 1880.38     386 1902.82   395.9 1910.12   399.2 1912.17
#Mann= 3 ,-1 , 0
       0     .12       0   215.5    .045       0   239.5     .12       0
Bank Sta=215.5,239.5
XS Rating Curve= 0 ,0
Exp/Cntr=0.3,0.1

Type RM Length L Ch R = 1 ,11221.6 ,245.1,250,251.1
XS GIS Cut Line= 3
     2099059.048      197483.835     2098991.808      197701.381
     2098944.897      197859.844
#Sta/Elev= 30
       0 1939.48     9.8 1935.12    22.8 1927.77    32.5 1924.69    35.8 1922.99
    48.8 1912.41    55.3 1904.31    61.8 1900.36   107.3 1876.02   123.6 1867.93
   156.1 1855.01   175.6 1846.12   178.9 1843.69   185.4 1837.19   191.9 1833.11
   201.7 1832.67   211.4 1830.83   221.2 1830.56   240.7 1830.23     2451830.527
   253.6 1831.66   263.3 1831.46   273.1 1835.45     286 1842.82     312 1860.44
   337.9 1874.51   350.8 1882.45   357.3 1886.83   363.8 1892.76     393 1909.14
#Mann= 3 ,-1 , 0
       0     .12       0   221.2    .045       0     245     .12       0
Bank Sta=221.2,245
XS Rating Curve= 0 ,0
Exp/Cntr=0.3,0.1

Type RM Length L Ch R = 1 ,10971.6 ,265.1,250,239.3
XS GIS Cut Line= 3
     2098873.405      197408.926     2098773.218      197586.179
      2098692.48      197814.553
#Sta/Elev= 30
       0 1948.89    12.9 1938.83    22.6 1932.46    29.1 1927.41    45.2 1918.55
    61.4 1911.52    87.3 1892.69      97 1887.16   100.2 1883.49   106.6 1873.37
   109.9 1868.86   113.1 1865.19   116.4 1862.74   145.4 1845.52   161.6 1832.22
   164.8 1830.56   168.1 1830.09   190.7 1828.22   206.9 1827.94   213.4 1828.26
   239.6 1833.82   259.2 1845.55   295.3 1865.43   324.7  1884.2   341.1 1891.38
   357.4 1899.94   373.8 1907.59   409.8 1920.09   426.2 1924.61   445.8 1928.92
#Mann= 3 ,-1 , 0
       0     .12       0   190.7    .045       0   213.4     .12       0
Bank Sta=190.7,213.4
XS Rating Curve= 0 ,0
Exp/Cntr=0.3,0.1

Type RM Length L Ch R = 1 ,10721.6 ,255,250,243.1
XS GIS Cut Line= 3
     2098493.573       197360.26     2098528.541      197572.058
     2098559.657      197825.296
#Sta/Elev= 30
       0 1971.65     9.8  1966.9    35.8 1950.98    68.3 1927.67    78.1 1918.34
    84.6 1913.39    94.3 1903.16   100.8    1898   110.6 1893.05   130.1 1881.03
   146.4 1868.29   162.6 1858.93   169.1 1853.65   172.4 1849.79   182.1 1834.03
   185.4    1831   195.2 1827.09   203.31825.841   221.2 1825.64     226 1825.71
   263.7 1831.57     303 1849.22   325.9 1862.87   335.7 1870.21   355.3  1880.2
   368.4 1888.97   381.5 1895.27   414.2 1908.87   433.8 1914.92   469.8 1923.87
#Mann= 3 ,-1 , 0
       0     .12       0   203.3    .045       0     226     .12       0
Bank Sta=203.3,226
XS Rating Curve= 0 ,0
Exp/Cntr=0.3,0.1

Type RM Length L Ch R = 1 ,10471.6 ,250.6,250,251.1
XS GIS Cut Line= 3
     2098196.087      197420.191     2098292.602      197653.094
     2098381.805      197852.368
#Sta/Elev= 30
       0 1964.35     6.6 1958.96    16.4  1956.8    19.6 1955.16    29.5 1945.63
    49.1 1931.04      72 1919.95    85.1 1907.63     108 1892.72   117.9 1883.57
   150.6 1862.65   160.4 1855.49   180.1 1845.82   206.3 1836.91   216.1 1826.12
   219.4 1824.23     239 1824.67   245.6 1823.84   261.9 1824.41   271.7 1826.89
   284.7 1826.93   291.2 1829.03   304.2 1837.86     314 1846.17   340.1 1864.42
   356.4 1873.56   382.4 1885.54   431.3 1905.84   454.1 1911.84   470.4 1914.42
#Mann= 3 ,-1 , 0
       0     .12       0     239    .045       0   261.9     .12       0
Bank Sta=239,261.9
XS Rating Curve= 0 ,0
Exp/Cntr=0.3,0.1

Type RM Length L Ch R = 1 ,10221.6 ,257.9,249.1,240.6
XS GIS Cut Line= 3
       2097950.9      197488.616     2098051.234      197709.953
     2098131.973      197921.638
#Sta/Elev= 30
       0 1963.25      13 1953.95    25.9 1946.38    29.2 1945.22    35.6 1944.32
    38.9  1942.7    51.8 1931.87      68 1921.11    77.8 1913.72    84.2 1906.43
     149 1861.88   168.5 1849.11   204.1 1829.31   213.8 1826.08   220.3  1823.3
   226.8 1821.48   230.1 1821.13   249.5 1821.45   262.4 1821.41   268.9 1822.99
   285.1  1824.3   291.6 1826.34     298 1832.28   333.6 1851.39     366 1871.08
   395.1 1886.51   401.6  1889.4   437.2 1897.31   459.9  1901.1   469.6  1901.9
#Mann= 3 ,-1 , 0
       0     .12       0   226.8    .045       0   249.5     .12       0
Bank Sta=226.8,249.5
XS Rating Curve= 0 ,0
Exp/Cntr=0.3,0.1

Type RM Length L Ch R = 1 ,9972.5  ,247.3,248.9,248.3
XS GIS Cut Line= 3
      2097672.49       197692.42     2097836.083      197831.923
     2097998.058      198008.645
#Sta/Elev= 30
       0 1910.99    26.1 1901.56    35.8  1895.9    55.4 1888.57    61.9 1883.96
    71.7 1873.83      88 1866.58   104.2 1856.91   123.8 1848.58   130.3 1844.26
   143.3 1838.68   169.4 1830.53   188.9 1821.82   195.4 1819.55   205.2 1817.38
   211.7 1816.84   234.4 1816.58   237.7 1816.56   240.9 1816.66   250.6 1819.86
   263.6 1820.42   270.1 1822.39   312.2 1841.98   341.3 1856.26   360.8 1867.21
     377 1877.78   383.4 1880.74   415.8 1890.67   428.8 1895.74   454.7 1900.75
#Mann= 3 ,-1 , 0
       0     .12       0   211.7    .045       0   234.4     .12       0
Bank Sta=211.7,234.4
XS Rating Curve= 0 ,0
Exp/Cntr=0.3,0.1

Type RM Length L Ch R = 1 ,9723.6  ,251.6,250,248.2
XS GIS Cut Line= 3
     2097511.427      197843.982      2097672.43      198010.246
      2097795.96      198139.952
#Sta/Elev= 30
       0 1941.23    29.3  1924.7    52.2  1913.9    55.4 1911.95    61.9 1906.59
    65.2 1905.06    71.7 1904.26    78.2 1902.22     101 1888.75   110.8 1884.33
   130.4 1867.85   133.6 1865.82   143.4 1861.11   146.7 1858.32   156.5  1848.6
     176  1834.2   192.3  1824.6   205.4 1818.42   211.9 1816.31     2201814.574
   224.9 1814.38   242.91814.416   257.5 1815.04   283.6 1820.77   293.3 1826.13
   312.9 1835.74   329.1 1845.64     365 1862.45   394.3 1873.76   410.6 1877.69
#Mann= 3 ,-1 , 0
       0     .12       0     220    .045       0   242.9     .12       0
Bank Sta=220,242.9
XS Rating Curve= 0 ,0
Exp/Cntr=0.3,0.1

Type RM Length L Ch R = 1 ,9473.6  ,249.1,250,250.7
XS GIS Cut Line= 3
     2097317.674      198026.306     2097495.851       198186.05
     2097610.863      198289.164
#Sta/Elev= 30
       0 1927.13    45.9 1899.08    49.2 1897.51    62.3 1893.55    78.7 1885.02
   104.9 1868.62   114.7 1861.52   124.6 1856.47   134.4 1849.53   150.8 1841.44
   173.7 1828.76   183.6  1824.5   196.7 1817.56   206.5 1813.89   213.1 1812.44
   227.81812.146   245.7 1812.04   250.81812.088   258.6 1812.16   261.8 1812.79
   277.9 1818.58   287.6 1820.62   297.2  1827.1   313.3 1836.34   316.5 1839.31
     323 1847.67   329.4 1851.25   351.9 1857.79   371.2 1859.04   393.8 1862.14
#Mann= 3 ,-1 , 0
       0     .12       0   227.8    .045       0   250.8     .12       0
Bank Sta=227.8,250.8
XS Rating Curve= 0 ,0
Exp/Cntr=0.3,0.1

Type RM Length L Ch R = 1 ,9223.6  ,247.7,250,251.4
XS GIS Cut Line= 3
     2097142.515      198191.132     2097311.673      198353.782
     2097430.666      198468.198
#Sta/Elev= 30
       0  1924.9     6.5 1920.79    16.3 1915.54    29.3 1906.71    35.8 1902.96
    48.9 1897.74    58.7 1892.34    81.5 1881.22     101 1873.64   114.1 1867.05
   130.4 1860.41   153.2 1847.53   156.4 1845.21   166.2 1835.33     176 1827.37
   192.3 1816.99   198.8 1814.07   208.6 1811.26   223.21809.269   228.2 1809.08
   246.21809.474   254.1 1811.19   263.8 1811.64     267 1812.33   283.2 1822.11
   299.4 1829.61   344.7 1847.19   364.1 1852.56  390.361857.165   399.8 1858.17
#Mann= 4 ,-1 , 0
       0     .12       0   223.2    .045       0   246.2     .12       0
  390.36     .06       0
Bank Sta=223.2,246.2
XS Rating Curve= 0 ,0
Exp/Cntr=0.3,0.1

Type RM Length L Ch R = 1 ,8973.6  ,247.8,248.5,249.5
XS GIS Cut Line= 3
     2096967.141      198333.579     2097134.148      198529.149
     2097242.739      198647.877
#Sta/Elev= 30
       0 1939.97    19.5 1926.14    35.8 1913.72    45.6 1905.58    61.8 1893.78
    74.9 1884.97    87.9  1877.3   133.5 1854.34   156.3 1844.69   169.3 1837.75
   185.6 1830.61   201.8 1821.09   211.6 1812.88   214.9 1811.16   218.1 1810.59
   227.9  1810.5   234.4 1809.67   245.61809.346   268.71809.048   279.7 1808.87
   289.4 1810.15   295.8 1811.63   308.7 1817.67   318.3 1820.31   344.1 1829.78
  354.47 1831.91   369.8 1833.65   382.7 1836.94   395.6 1838.94   418.1 1840.11
#Mann= 4 ,-1 , 0
       0     .12       0   245.6    .045       0   268.7     .12       0
  354.47     .06       0
Bank Sta=245.6,268.7
XS Rating Curve= 0 ,0
Exp/Cntr=0.3,0.1

Type RM Length L Ch R = 1 ,8725.1  ,246.1,250,250.5
XS GIS Cut Line= 3
     2096777.124      198477.582     2096960.032        198701.9
     2097059.487      198823.087
#Sta/Elev= 30
       0 1905.96    16.3 1900.15    48.8 1884.37    68.3 1873.58    87.8 1864.59
   126.8 1849.73   146.3 1841.01   159.4 1838.08   169.1 1834.95   178.9 1831.01
   198.4 1821.44   217.9 1808.93   221.1 1808.04   237.4 1809.42   250.4 1809.68
   269.9 1808.59  275.271807.411   279.7 1806.39   286.2 1806.14   292.7 1806.24
   299.2 1807.36     309  1808.9   312.3 1810.27     358 1832.55  366.891835.819
   380.9 1840.08   397.2 1841.66  411.061846.552  435.421852.761   446.2 1854.71
#Mann= 6 ,-1 , 0
       0     .12       0  275.27    .045       0   299.2     .12       0
  366.89    .016       0  411.06     .06       0  435.42     .12       0
Bank Sta=275.27,299.2
XS Rating Curve= 0 ,0
Exp/Cntr=0.3,0.1

Type RM Length L Ch R = 1 ,8475.1  ,241.2,242.5,246.4
XS GIS Cut Line= 3
     2096614.216      198601.042     2096737.469      198814.246
     2096877.342      198997.238
#Sta/Elev= 30
       0 1861.59    38.9 1848.79   56.67 1841.99    71.3 1837.64    90.7  1832.9
   129.6 1824.27  141.381822.144     162 1818.01   186.81814.123   200.9 1812.11
   210.6 1809.25  220.361807.754   239.8 1804.81   246.3 1804.64  260.411804.812
   265.7 1805.68   272.2 1807.76   278.7 1808.11     282 1808.93   294.9 1813.19
  317.871819.352  327.491823.875   343.6 1831.07   359.8 1834.07   369.5 1837.96
  375.981839.894   398.7 1843.26   431.2 1845.79   450.6 1845.75   476.6  1844.9
#Mann= 10 ,-1 , 0
       0     .12       0   56.67     .06       0  141.38     .12       0
   186.8    .016       0  220.36     .12       0   239.8    .045       0
  260.41     .12       0  317.87     .06       0  327.49    .016       0
  375.98     .06       0
Bank Sta=239.8,260.41
XS Rating Curve= 0 ,0
Exp/Cntr=0.3,0.1

Type RM Length L Ch R = 1 ,8232.6  ,223.3,232.5,240.3
XS GIS Cut Line= 2
     2096403.381      198663.532     2096675.179      199190.529
#Sta/Elev= 30
       0 1904.37    26.2 1886.17    68.8 1858.52    78.6 1851.52   108.1  1837.1
   124.5 1830.49  136.131827.014   157.2 1821.16   173.6 1817.68     226 1809.21
   252.2 1806.72  281.411807.239   288.3 1807.34  314.341805.082  320.151804.536
     321  1804.4   330.9 1803.37  345.071804.432   357.1  1807.8   366.9 1808.08
   380.41809.991     416 1814.98  432.991816.463  499.461824.448  505.771825.289
   520.9 1828.45   537.3 1830.12  565.941835.657  578.651838.083     593 1839.13
#Mann= 13 ,-1 , 0
       0     .12       0  136.13     .06       0  281.41    .016       0
  314.34     .12       0  320.15    .016       0     321    .045       0
  345.07    .016       0   380.4     .06       0  432.99     .12       0
  499.46     .06       0  505.77    .016       0  565.94     .06       0
  578.65     .08       0
Bank Sta=321,345.07
XS Rating Curve= 0 ,0
Exp/Cntr=0.3,0.1

Type RM Length L Ch R = 1 ,8000.2  ,574.8,558.8,541.3
XS GIS Cut Line= 4
     2096238.918      198685.227     2096319.167      198880.115
     2096351.719      199184.803     2096508.221      199331.024
#Sta/Elev= 30
       0 1921.95    19.5 1906.13    35.7 1896.07    51.9 1883.65    64.8 1872.29
    90.8 1855.06   100.5 1850.88   142.7 1838.96  167.611829.276   188.1 1822.77
   223.8 1813.94  245.58    1807   253.1 1805.63     302 1805.14   318.21803.995
   334.6 1802.99   341.2 1804.16   347.7 1806.76  352.881806.646     364 1805.84
  441.73 1807.26  498.771809.129  537.461813.755  546.631814.351  607.621819.308
   631.41821.336  658.411822.487   689.2 1826.43   718.4 1833.52   731.4 1835.54
#Mann= 13 ,-1 , 0
       0     .12       0  167.61     .06       0  245.58     .12       0
   318.2    .045       0   341.2     .12       0  352.88     .06       0
  441.73     .08       0  498.77     .06       0  537.46     .12       0
  546.63    .016       0  607.62     .12       0   631.4    .016       0
  658.41     .06       0
#XS Ineff= 2 , 0
                          459.03         1811.82
Permanent Ineff=
       F       F
Bank Sta=318.2,341.2
XS Rating Curve= 0 ,0
Exp/Cntr=0.3,0.1

Type RM Length L Ch R = 1 ,7441.4  ,329.3,325.3,321.4
XS GIS Cut Line= 2
     2095687.121      198981.446     2096285.701       199514.76
#Sta/Elev= 30
       0 1935.56    49.1 1934.85   70.481931.455    78.5 1928.62    94.9 1919.07
   130.9 1894.91   140.7 1885.35   150.5 1879.13   153.8 1876.21   189.8 1842.01
   212.7 1825.22   225.8 1814.44   235.6 1803.83   238.9 1801.11   245.4 1799.07
     252 1798.87   268.3 1799.02   281.4  1801.4  304.79 1801.44   382.8 1802.86
   664.3 1802.95   687.2 1805.98   710.1 1818.03   723.2 1820.68  750.121829.148
   762.4 1835.28   778.8 1837.15   785.3 1842.16     7951846.052   801.7 1848.73
#Mann= 7 ,-1 , 0
       0     .06       0   70.48     .12       0   245.4    .045       0
   268.3     .12       0  304.79     .06       0  750.12    .016       0
     795     .12       0
#XS Ineff= 2 , 0
                          554.18         1808.11
Permanent Ineff=
       F       F
Bank Sta=245.4,268.3
XS Rating Curve= 0 ,0
Exp/Cntr=0.3,0.1

Type RM Length L Ch R = 1 ,7116    ,443.4,436.1,427.3
XS GIS Cut Line= 2
     2095380.239      199221.002     2096066.562      199647.694
#Sta/Elev= 30
       0 1865.38    13.1 1870.72    26.2 1872.94      36 1878.34    52.4 1883.75
    91.6 1894.37     108 1898.16   130.9 1899.75   147.2 1891.41   199.6 1852.79
   225.8 1831.47   235.6 1820.33   245.4 1811.07   258.5 1801.35     265 1799.36
   297.7 1800.56   323.9 1798.01   343.6 1797.46   350.1 1798.12   356.6 1800.22
  377.36 1800.07   477.7 1799.07   575.8 1800.46   677.3 1799.75   696.9 1802.74
   729.6 1815.32  772.231826.198   785.2 1829.62   801.6  1830.3   808.2 1834.21
#Mann= 5 ,-1 , 0
       0     .12       0   323.9    .045       0   350.1     .12       0
  377.36     .06       0  772.23    .016       0
#XS Ineff= 2 , 0
                          603.72          1805.3
Permanent Ineff=
       F       F
Bank Sta=323.9,350.1
XS Rating Curve= 0 ,0
Exp/Cntr=0.3,0.1

Type RM Length L Ch R = 1 ,6680    ,620.4,635,633.8
XS GIS Cut Line= 3
     2095159.196      199620.799     2095761.658      199739.924
      2095884.46      199999.073
#Sta/Elev= 30
       0 1848.19    42.5 1838.16     1061820.854   117.6 1818.54   124.1 1814.97
   130.7 1812.58   156.8 1807.93  166.261805.545   192.7 1802.54     196 1801.32
   202.5 1795.93   205.8 1795.13   222.1 1794.84   231.9 1795.03     245 1795.54
   258.1 1797.42  296.371797.747   467.1 1797.15   552.1 1799.36   617.4 1799.96
  736.56 1807.41   760.8 1810.81   773.8 1811.16   777.1 1811.99  794.551823.057
     826 1842.42   835.7 1852.29     839 1854.44   871.6 1872.03   900.9 1884.95
#Mann= 8 ,-1 , 0
       0     .12       0     106     .06       0  166.26     .12       0
   205.8    .045       0   231.9     .12       0  296.37     .06       0
  736.56    .016       0  794.55     .12       0
Bank Sta=205.8,231.9
XS Rating Curve= 0 ,0
Exp/Cntr=0.3,0.1

Type RM Length L Ch R = 1 ,6045    ,384.4,383.8,382.2
XS GIS Cut Line= 2
     2095095.747      199814.117     2095569.705      200292.137
#Sta/Elev= 30
       0 1832.43    19.6 1822.85   38.18 1817.16    71.9 1808.88  122.981804.491
  191.111802.311   264.7 1800.99   303.9 1797.78   333.3 1793.66  358.481793.106
   370.21791.657   385.6 1791.02   393.91791.583   405.2 1794.28     4191793.962
  472.411793.554  537.961796.639     562 1797.34   568.6 1799.62  573.451803.121
   581.7 1810.02   584.9 1811.64   594.7  1812.5     598 1814.37   607.8 1823.94
  619.16 1837.23   637.2 1855.11     647  1863.6   656.8 1869.28   673.2 1875.85
#Mann= 12 ,-1 , 0
       0     .12       0   38.18     .06       0  122.98     .12       0
  191.11     .06       0  358.48     .12       0   370.2    .045       0
   393.9     .06       0     419    .016       0  472.41     .06       0
  537.96     .12       0  573.45    .016       0  619.16     .12       0
Bank Sta=370.2,393.9
XS Rating Curve= 0 ,0
Exp/Cntr=0.3,0.1

Type RM Length L Ch R = 1 ,5661.2  ,472.7,455,435.7
XS GIS Cut Line= 3
     2094896.609      200172.498      2095252.76      200470.176
     2095399.223      200459.715
#Sta/Elev= 30
       0 1817.32     6.5 1813.85    32.7 1804.17      49  1798.6   59.25 1796.39
   104.6 1792.48   156.9 1791.53   264.8 1792.24     268  1792.1  273.571789.664
  276.241788.883   284.4 1788.57   300.7 1788.97   307.51790.519   313.8 1792.04
   320.3 1795.36   323.6 1796.12  337.251797.042     438 1804.78   454.4 1807.72
  461.481807.865   480.5 1807.82   490.3 1811.79  495.241813.027  519.721818.797
  562.771819.505   575.1 1819.44   578.4 1820.17   594.7 1826.91     611 1831.29
#Mann= 11 ,-1 , 0
       0     .12       0   59.25     .06       0  273.57     .08       0
  276.24    .045       0   300.7     .08       0   307.5     .06       0
  337.25     .08       0  461.48    .016       0  495.24     .06       0
  519.72     .08       0  562.77     .06       0
Bank Sta=276.24,300.7
XS Rating Curve= 0 ,0
Exp/Cntr=0.3,0.1

Type RM Length L Ch R = 1 ,5206.2  ,227.8,228.7,231.3
XS GIS Cut Line= 2
      2094748.35      200679.372     2095369.628      200609.663
#Sta/Elev= 30
       0  1844.1     6.6 1843.87    22.9 1840.32    49.1 1836.52    65.5 1832.99
    75.3 1829.97    85.1  1825.3   111.3 1811.28   117.8 1807.16   124.4 1802.36
   130.9 1795.62   134.2 1791.62   137.5 1788.82  140.361787.572     144 1787.17
   166.9 1787.53   170.2  1787.8     180 1790.04   340.4  1794.7   366.6 1796.06
   438.6 1798.14  483.881801.107   487.7 1801.34   497.5 1803.93   500.8 1804.28
   543.4 1804.84   576.1 1806.47   602.3 1810.15  624.38 1812.32   625.2 1812.38
#Mann= 5 ,-1 , 0
       0     .12       0  140.36    .045       0   166.9     .06       0
  483.88    .016       0  624.38     .06       0
Bank Sta=140.36,166.9
XS Rating Curve= 0 ,0
Exp/Cntr=0.3,0.1

Type RM Length L Ch R = 1 ,4977.5  ,455.2,462.3,469.7
XS GIS Cut Line= 3
     2094734.171      200904.021     2094929.404      200887.905
     2095293.212      200891.893
#Sta/Elev= 30
       0 1844.28   12.651841.327    32.6 1838.91   49.311833.205    55.5 1830.05
    84.9  1818.1    91.4 1816.52  103.531815.602   120.8 1812.84   133.9 1808.91
   143.7 1806.89   150.2 1803.12     160 1793.84   163.2  1791.4   166.5 1789.74
     173 1787.37   186.1 1787.39   202.4 1786.62  210.911787.375   218.8 1789.81
   235.2  1789.3  251.311789.649   353.2 1790.62   392.6 1792.81  428.551795.806
   458.1 1799.52  487.641804.963   500.7 1805.12  508.141806.643   559.7 1811.46
#Mann= 11 ,-1 , 0
       0     .06       0   12.65     .12       0   49.31     .06       0
  103.53     .12       0   186.1    .045       0  210.91     .06       0
  251.31    .016       0  428.55     .06       0   458.1     .08       0
  487.64    .016       0  508.14     .06       0
Bank Sta=186.1,210.91
XS Rating Curve= 0 ,0
Exp/Cntr=0.3,0.1

Type RM Length L Ch R = 1 ,4515.2  ,458.1,473.5,483
XS GIS Cut Line= 2
     2094651.299      201172.552     2095231.172      201394.667
#Sta/Elev= 30
       0 1864.19    29.4 1842.16    52.3 1827.02    68.6 1818.03    91.5 1809.13
   143.8 1796.03   160.1 1793.05   196.1 1787.51  217.851787.501   264.7 1788.48
  322.711788.445   349.7 1788.45   362.8 1787.03     366 1786.21   375.8 1785.49
   382.11784.311   385.6 1784.14   406.1 1784.23   437.9 1784.24   444.5 1784.84
     451 1787.93   457.6 1789.26  505.841805.767   516.4 1810.16   529.4 1811.44
   532.7 1812.78   542.5 1818.48   565.4 1829.69   578.5 1837.03     621 1855.59
#Mann= 7 ,-1 , 0
       0     .12       0  217.85     .06       0  322.71     .12       0
   382.1    .045       0   406.1     .12       0  505.84    .016       0
   542.5     .12       0
#XS Ineff= 2 , 0
          262.23 1791.66
Permanent Ineff=
       F       F
Bank Sta=382.1,406.1
XS Rating Curve= 0 ,0
Exp/Cntr=0.3,0.1

Type RM Length L Ch R = 1 ,4041.7  ,470.7,474.7,477.9
XS GIS Cut Line= 2
     2094519.913      201357.026     2094960.289      201826.645
#Sta/Elev= 30
       0 1907.21    22.9 1889.69      85 1844.95   104.6 1829.91   114.4  1820.4
   137.3 1803.15   156.9 1790.71  167.911785.993   186.3 1784.35   225.5 1785.69
   287.6 1785.91   303.9  1784.1   330.1 1784.98   343.1 1783.65  398.561784.974
   428.1 1785.44     4491782.806   464.1 1782.33   473.11783.406   483.7 1793.24
   490.2    1797   503.3  1802.5  519.851807.527   539.2 1813.95  550.021816.331
   565.4 1816.46   575.2 1824.12  581.351826.456   620.9 1837.54   643.8  1845.2
#Mann= 8 ,-1 , 0
       0     .12       0  167.91     .06       0  398.56     .12       0
     449    .045       0   473.1     .12       0  519.85     .06       0
  550.02    .016       0  581.35     .12       0
Bank Sta=449,473.1
XS Rating Curve= 0 ,0
Exp/Cntr=0.3,0.1

Type RM Length L Ch R = 1 ,3567    ,287.1,289.8,292
XS GIS Cut Line= 2
     2094333.835      201492.233     2094685.114      202029.383
#Sta/Elev= 30
       0 1882.03    26.2 1867.34    42.6 1854.83    65.5 1840.33      72 1837.61
    85.1 1834.95    98.2 1829.88   117.9 1825.47   124.4 1822.85   150.6 1806.35
   173.6 1794.02  185.621785.295   193.2 1780.44   212.8 1780.08   216.1 1780.28
  220.92 1781.86   245.6 1781.25   271.8 1782.99   324.2 1782.51   415.9 1785.14
   445.3 1787.22  486.181794.611   517.4 1797.07     537 1796.04   586.2 1810.01
   605.8 1812.49  609.171814.026   615.6 1816.31   635.3 1816.46   641.8  1820.7
#Mann= 7 ,-1 , 0
       0     .12       0  185.62     .08       0   193.2    .045       0
   216.1     .08       0  220.92     .06       0  486.18     .12       0
  609.17    .016       0
Bank Sta=193.2,216.1
XS Rating Curve= 0 ,0
Exp/Cntr=0.3,0.1

Type RM Length L Ch R = 1 ,3277.2  ,311.1,314.2,315.7
XS GIS Cut Line= 2
     2094099.641      201603.934     2094400.685      202197.062
#Sta/Elev= 30
       0 1846.76    16.4 1840.13    39.3 1832.61    91.8 1817.93  113.521811.008
  120.151809.042   140.9    1804   157.3  1797.4   173.7 1788.71   183.5 1781.21
   186.8 1780.15   196.6 1781.09     2101779.893   226.1 1778.89   234.31779.712
   242.5  1780.8  257.141780.539   265.4  1781.6   285.1  1779.6     308 1778.54
  326.421780.578   370.3 1781.63   452.2 1781.01  462.631782.665   468.6 1783.91
   481.7 1783.91  518.671793.481   550.5 1799.31   612.7 1814.36   665.2 1823.63
#Mann= 9 ,-1 , 0
       0     .12       0  113.52     .06       0  120.15     .12       0
     210    .045       0   234.3     .06       0  257.14     .12       0
  326.42     .06       0  462.63     .12       0  518.67     .06       0
#XS Ineff= 2 , 0
                          470.28         1785.41
Permanent Ineff=
       F       F
Bank Sta=210,234.3
XS Rating Curve= 0 ,0
Exp/Cntr=0.3,0.1
